--- RattlesnakeRun.prj (project) ---

Proj Title=Basic Project File
Current Plan=p01
Default Exp/Contr=0.3,0.1
English Units
Geom File=g01
Flow File=f01
Plan File=p01
Y Axis Title=Elevation
X Axis Title(PF)=Main Channel Distance
X Axis Title(XS)=Station
BEGIN DESCRIPTION:
END DESCRIPTION:
DSS File=dss
DSS Export Rating Curves= 0
DSS Export Rating Curve Sorted= 0
DSS Export Volume Flow Curves= 0
DXF OffsetX= 0
DXF OffsetY= 0
DXF ScaleX= 1
DXF ScaleY= 10

--- RattlesnakeRun.p01 (plan) ---

Plan Title=Basic Plan File
Short Identifier=Basic Plan File
Geom File=g01
Flow File=f01
Subcritical Flow
K Sum by GR= 0
Std Step Tol= 0.01
Critical Tol= 0.01
Num of Std Step Trials= 20
Max Error Tol= 0.33
Flow Tol Ratio= 0.001
Split Flow NTrial= 30
Split Flow Tol= 0.02
Split Flow Ratio= 0.02
Log Output Level= 0
Friction Slope Method= 1
Unsteady Friction Slope Method= 2
Calc Critical at every XS
Parabolic Critical Depth
Global Vel Dist= 0 , 0 , 0
Global Log Level= 0
CheckData=True
Encroach Param=-1 ,0,0, 0
Computation Interval=1HOUR
Output Interval=1HOUR
Run HTab= 0
Run UNet= 0
Run PostProcess= 0
UNET Theta= 1
UNET ZTol= 0.02
UNET ZSATol= 0.1
UNET MxIter= 20
UNET MaxInSteps= 20
UNET DtIC= 0
UNET DtMin= 0
UNET MaxCRTS= 20
UNET WFStab= 2
UNET SFStab= 1
UNET WFX= 1
UNET SFX= 1
UNET Convert EG Bridges=-1
UNET Use Existing IB Tables=-1
Instantaneous Interval=1HOUR
DSS File=dss
Write IC File= 0
Write Velocity= 0
Write Detailed= 0

--- RattlesnakeRun.f01 (steady flow) ---

Flow Title=Basic Flow File
Program Version=4.10
Number of Profiles= 1
Profile Names=P1
River Rch & RM=RattlesnakeRun,Reach1          ,31588.56
    1036
River Rch & RM=RattlesnakeRun,Reach1          ,18597.36
    2225
Boundary for River Rch & Prof#=RattlesnakeRun,Reach1          , 1
Up Type= 0
Dn Type= 3
Dn Slope=0.01133
DSS Import GetInterval= 0
DSS Import GetPeak= 0
DSS Import FillOption= 0

--- RattlesnakeRun.g01 (geometry) ---

Geom Title=Generated by CreateGeometryFile written by the GeoFIRM tool.
Program Version=4.10

River Reach=RattlesnakeRun  ,Reach1
Reach XY= 30
2442916.88672319330849.485862434 2444616.9735461330101.742935359
2444722.52910927330464.2428665162445403.77905911330522.923523441
2446546.63602535331409.1874989422446959.12109278 330804.61488919
2447636.56068277330920.0510100132447731.12217344330659.847134098
2448536.75310811330942.1884329322449852.80985919329992.278259277
2450449.59803569 329979.691342192451329.50244386329354.170611605
 2451942.8706397329198.0941521082453965.52669936329944.882356688
2454761.53363752330332.9898481822455505.80445869 331655.38582544
2456125.94331028 331981.913715692456166.04756078332856.392609775
2457055.37058528335215.3337580262456916.68451095335906.553832263
2457075.33576845336584.2572012692456722.03726244336784.344071433
2456475.00593236337316.7573766862456674.22469403337741.236514598
2457005.82179986337775.9585580232457124.74544652338520.750375524
 2458535.3358012339721.2712684422460017.90403028339131.267199099
2461314.23575519339104.3017018592462317.54083519339566.844083861

Type RM Length L Ch R = 1 ,31588.56,1014.718,1010.728,1001.757
XS GIS Cut Line= 3
2443110.15175661331316.4691804352442918.77156194330849.163028434
2442728.57049878330384.737120017
#Sta/Elev= 30
       0  502.32   55.74  498.44  177.07  491.68  245.93  484.47  301.67  479.75
  383.65  470.99   439.4  468.34  462.35  468.03  472.19  468.63  482.02  467.85
  491.86   468.6  494.87  468.24   501.7  466.36  504.98  466.26  514.66  468.49
  521.38  468.85  547.62  468.33   583.7  469.86  652.58  470.91  688.67  472.43
  750.99  477.54  780.51  481.33  806.75  482.85  819.87  482.85  839.55  485.74
  852.67  486.16  898.59   491.3  921.55  493.26   980.6  496.69 1006.84  497.44
#Mann= 3 , 0 , 0
       0     .12       0  494.87    .045       0  514.66     .12       0
Bank Sta=494.87,514.66
XS Rating Curve= 0 ,0
Exp/Cntr=0.3,0.1

Type RM Length L Ch R = 1 ,31083.15,493.9902,494.6823,494.9896
XS GIS Cut Line= 4
    2443635.6074    331186.48552   2443365.16109    330625.68677
    2443136.3059     330178.1729   2442748.02059    329637.00633
#Sta/Elev= 30
  -622.6   482.6  -524.3  480.12  -439.1  474.21  -353.9  470.47 -252.32  469.94
 -101.58  465.55   -9.99  465.86   -3.28  465.62    3.26  464.11      10  465.39
  130.55  465.12  159.93   468.3  169.72  466.26  264.37   467.8   270.9  467.55
  280.69  465.53  303.54  467.83  594.06   471.7  639.76  472.69  669.15  474.47
  796.48  474.86  819.34   475.7   887.9  482.33  914.02  486.45  930.35  486.96
   953.2  489.74  985.85  491.12 1021.77  496.15 1129.51  502.41 1168.69  500.55
#Mann= 3 ,-1 , 0
  -622.6     .12       0   -9.99    .045       0      10     .12       0
#XS Ineff= 2 , 0
                           158.8          470.37
Permanent Ineff=
       F       F
Bank Sta=-9.99,10
XS Rating Curve= 0 ,0
Exp/Cntr=0.3,0.1

Type RM Length L Ch R = 1 ,30588.47,875.2925,912.1952,916.5176
XS GIS Cut Line= 5
   2444134.75666    331616.05159   2443999.65523    330818.11814
     2443800.424    330400.34864   2443585.09569    329948.82559
   2443350.03448    329723.69054
#Sta/Elev= 30
-1272.13  480.63-1180.39  481.58 -1137.8  480.62-1055.89  480.78 -892.06  471.14
 -790.49  469.23 -711.86  469.65 -610.29  473.04 -528.37  472.49 -449.81  469.88
 -404.17  469.52 -316.17  472.62 -277.05  472.15 -250.98  472.96  -153.2  463.93
  -48.89  460.83  -13.04  461.58   -3.26  459.56    6.54  461.58   117.7   461.8
  140.59   460.9  209.25  462.15  313.88  460.62  519.77  463.29  594.63  465.96
  653.22  470.05  721.57  478.54  773.65  482.68   812.7  483.88  825.72  483.37
#Mann= 3 , 0 , 0
-1272.13     .12       0  -13.04    .045       0    6.54     .12       0
#XS Ineff= 2 , 0
                          413.45          464.09
Permanent Ineff=
       F       F
Bank Sta=-13.04,6.54
XS Rating Curve= 0 ,0
Exp/Cntr=0.3,0.1

Type RM Length L Ch R = 1 ,30067.16,357.81,390.89,391.52
XS GIS Cut Line= 5
2444231.75515644331313.1607881042444437.59956102 330683.20765169
2444266.52345961330166.4524516022444196.06690761329954.975840434
2444325.07124278329646.494173944
#Sta/Elev= 30
       0  480.68   26.12  481.18   58.76  480.19   81.62  479.01  130.59  474.95
  186.09  471.88   323.2  466.13  424.41  463.11  502.76  463.07  587.64  463.99
  633.35  464.82  662.73  466.57  829.97  461.24 1043.11  460.74 1125.09  459.38
 1167.72  457.92 1180.84  458.62 1191.28  458.03 1197.23  457.68 1211.16  457.94
 1279.19  458.59 1308.69  460.37 1328.36  462.37 1370.97  468.69  1426.7   472.9
 1551.27  483.83 1597.16  486.97 1649.61  489.23 1698.78  488.54 1764.34  489.93
#Mann= 3 , 0 , 0
       0     .12       0 1191.28    .045       0 1211.16     .12       0
Bank Sta=1191.28,1211.16
XS Rating Curve= 0 ,0
Exp/Cntr=0.3,0.1

Type RM Length L Ch R = 1 ,29676.27,584.5273,587.8048,574.9554
XS GIS Cut Line= 5
    2444367.6417    331780.64935    2444482.2248    330553.21874
   2444600.79084    330121.56245   2444856.55443    329687.26575
   2444761.73868    329370.92714
#Sta/Elev= 30
-1703.93  488.92-1628.52  485.53-1553.11  477.78 -1494.1  478.94-1395.74  470.85
-1346.56   471.1-1274.43  474.76-1215.41  470.56-1166.23  471.63-1113.78  469.89
-1061.32  465.23 -989.19   463.7 -779.36  463.77 -595.75  467.49 -471.16  466.68
 -376.41  461.03  -10.99  456.71   -3.88  455.66   10.15  456.97   45.21  457.88
   97.57   463.9  143.39  465.92  195.76  471.69  257.94  474.37  352.85  473.89
  408.49   479.1  670.14  496.36  683.22   495.1  758.42  497.78  810.74  496.52
#Mann= 3 ,-1 , 0
-1703.93     .12       0  -10.99    .045       0   10.15     .12       0
Bank Sta=-10.99,10.15
XS Rating Curve= 0 ,0
Exp/Cntr=0.3,0.1

Type RM Length L Ch R = 1 ,29088.47,512.5273,516.5768,512.5553
XS GIS Cut Line= 4
   2444789.56703    330836.08924   2444893.83093    330484.41048
   2445024.40613    330043.98419   2445581.18323    329648.70513
#Sta/Elev= 30
 -366.81  477.21 -311.13  477.52 -193.23  471.26 -176.85  469.72 -163.75  465.68
  -144.1  461.81 -124.45  460.48  -85.15   455.6  -55.68  453.76  -10.27  454.28
       0  452.82    9.71  454.49   87.97  457.79  166.16  457.19  228.06  459.29
  351.86  461.29  400.73  464.01  478.98  471.44  518.18  473.73  642.33   474.9
  782.82  478.22  841.62  482.87  851.43  484.14  857.96  486.52  867.76  487.39
  916.77  488.57  926.57  492.42  982.11  493.68 1086.66  498.61  1142.2  499.41
#Mann= 3 ,-1 , 0
 -366.81     .12       0  -10.27    .045       0    9.71     .12       0
Bank Sta=-10.27,9.71
XS Rating Curve= 0 ,0
Exp/Cntr=0.3,0.1

Type RM Length L Ch R = 1 ,28597.49,961.8607,992.4432,1014.874
XS GIS Cut Line= 3
2445277.87248677331261.6418622732445357.48486036330499.537415355
2445409.70194753330002.634209692
#Sta/Elev= 30
       0  477.92   72.04  475.38  157.18  470.57  239.04  463.69  317.63  459.74
  363.48  459.36  438.79  456.58  501.01  455.44  510.83  456.11  589.42  455.91
  635.27  456.77  651.64  455.02  690.94   452.7  713.86  452.01  726.96  452.54
  734.72  451.52  740.05  450.52  754.34  452.61  841.36  453.47  857.69  455.75
  887.08  455.75  909.94  458.02  945.86  457.72  981.78  459.25 1001.37  461.27
 1014.44  463.63 1050.36  467.15 1177.72  478.36 1223.44  483.61 1265.89  486.43
#Mann= 3 , 0 , 0
       0     .12       0  734.72    .045       0  754.34     .12       0
Bank Sta=734.72,754.34
XS Rating Curve= 0 ,0
Exp/Cntr=0.3,0.1

Type RM Length L Ch R = 1 ,28088.47,530.1951,529.7515,521.5281
XS GIS Cut Line= 3
   2445365.55834    331282.03848   2445698.06489     330863.9212
    2446051.6695    330421.27445
#Sta/Elev= 30
 -534.21  479.75 -481.77  477.92 -426.06  474.06 -357.23  467.85 -311.35  462.21
 -285.13  460.21 -193.37   455.8 -134.37  454.76  -81.93  451.19  -32.77  449.82
  -13.11  448.29       0  447.78    8.69  448.44   16.37  449.74   81.87  449.64
  157.19  453.67  173.57   453.5  203.04  455.38  235.79  455.88  245.61   456.8
  258.71  456.43  288.18  458.25  314.38  461.21  327.48  459.32  347.13  459.21
  366.78  464.65  386.43  466.97  438.83  471.36  501.05  473.98  566.54  479.03
#Mann= 3 , 0 , 0
 -534.21     .12       0  -13.11    .045       0    8.69     .12       0
Bank Sta=-13.11,8.69
XS Rating Curve= 0 ,0
Exp/Cntr=0.3,0.1

Type RM Length L Ch R = 1 ,27558.72,487.0486,470.2485,448.1023
XS GIS Cut Line= 3
   2445816.62436    331674.44583   2446062.24034    331238.62846
   2446312.94194    330793.78748
#Sta/Elev= 30
 -562.79  478.38  -530.1  477.95 -484.32  476.06 -271.79  463.98 -239.09  463.21
 -229.28  463.65 -222.74  462.13 -212.93  456.83 -209.66  455.85 -150.81  453.54
 -144.27  452.08  -108.3  449.18  -55.98  447.52  -23.25  447.58   -16.7  447.16
   -9.99  445.87    -.34  444.97   10.01  446.04   29.12  448.98   38.94  448.05
   61.85   449.7   94.59  450.74  182.96  451.63  271.34  453.56  317.17  456.74
  323.71  457.89  343.35   459.7  362.99  462.82  415.36  466.15  448.09  466.32
#Mann= 3 ,-1 , 0
 -562.79     .12       0   -9.99    .045       0   10.01     .12       0
Bank Sta=-9.99,10.01
XS Rating Curve= 0 ,0
Exp/Cntr=0.3,0.1

Type RM Length L Ch R = 1 ,27088.47,507.21,480.48,445.47
XS GIS Cut Line= 5
2446598.45744403 332046.491342442446484.05544186331603.105746269
2446492.90745828 331404.283637362446517.90970486331216.387031525
2446384.50905302330733.773495436
#Sta/Elev= 30
       0  468.08   68.69  467.62  160.27   465.8  242.04  465.28  327.08     463
  343.43  461.94   369.6  456.66  389.22  455.15  454.64  452.42  484.01  451.97
   519.9  448.44  588.41  445.85  634.09   445.2  643.88   444.7  646.85   443.8
  653.66  442.06  667.14  443.66   679.8  444.27  692.88   443.8  709.22  444.51
  735.36  444.53  784.38  445.88  859.57  445.53  882.48  447.28   928.3     448
  944.66  449.59  977.38  449.69 1052.66  451.98 1235.92  465.03 1347.19  471.22
#Mann= 3 ,-1 , 0
 -650.82     .12       0  -10.03    .045       0   10.02     .12       0
Bank Sta=646.85,667.14
XS Rating Curve= 0 ,0
Exp/Cntr=0.3,0.1

Type RM Length L Ch R = 1 ,26607.99,1471.443,1560.969,1625.222
XS GIS Cut Line= 4
2447125.02430427331704.0533790142446979.82938468331256.745874688
2446783.80713893331101.8925098482446435.84622069330827.010513693
#Sta/Elev= 30
       0  464.78   22.86  462.67   81.65  459.56  156.76  457.77  192.69   455.6
  300.46  457.47  349.45   454.8  476.77  452.22  570.85  447.81  580.59  446.47
  609.79  444.71  687.85  441.39  694.14  440.95  700.63  439.04  708.16  439.86
  716.85   440.7  746.18   440.3  817.91  444.18  879.86  444.78  918.99   446.2
  935.29  447.35  951.59  450.07  980.94  451.21  990.72  455.92  1000.5  457.71
 1023.32  457.74 1059.19  460.74  1124.4  463.77 1143.97  465.63 1163.53  465.66
#Mann= 3 , 0 , 0
       0     .12       0  687.85    .045       0  708.16     .12       0
Bank Sta=687.85,708.16
XS Rating Curve= 0 ,0
Exp/Cntr=0.3,0.1

Type RM Length L Ch R = 1 ,26057.4 ,491.59,468.93,439.39
XS GIS Cut Line= 5
2447196.44017194331622.1283460262447003.06227785330937.950908601
2447126.01478785330816.9019381112447185.35390803330763.992595106
2447057.15272085330261.008692935
#Sta/Elev= 30
       0  456.85   58.98  455.04  186.76  453.24  252.28   453.9  330.92  449.05
  353.85  448.17  386.62  447.36  429.21  448.24  452.14  447.79  540.61  441.92
  701.15  440.72  795.62  437.63  831.43  436.95  857.48  437.45  863.99   437.1
  872.96  435.37  877.01  435.21  892.95  437.43  912.14  438.94   934.4  442.19
  963.02   442.7  982.61  445.09 1011.99  447.56 1054.43  448.02 1109.93  446.56
 1220.92  448.83  1305.8  452.67 1393.94  458.03 1429.85  460.94 1482.09  462.56
#Mann= 3 , 0 , 0
       0     .12       0  872.96    .045       0  892.95     .12       0
Bank Sta=872.96,892.95
XS Rating Curve= 0 ,0
Exp/Cntr=0.3,0.1

Type RM Length L Ch R = 1 ,25588.47,984.1338,1000,953.161
XS GIS Cut Line= 3
   2447588.68315    331818.69619    2447554.3325    330927.41615
   2447528.63078    330270.83282
#Sta/Elev= 30
 -891.94  460.28 -783.73  458.22 -711.59  459.65 -678.79  459.64 -580.42  457.24
 -534.51  455.14 -377.11   449.7 -141.01  436.22 -114.77  435.35 -101.66  435.73
  -91.82  434.58  -81.98  431.85  -75.42  431.23  -39.35  431.14  -32.79  432.46
  -26.23  435.25  -22.95  435.11   -9.98  430.75   -3.28  429.96    6.54  430.78
    9.81  431.77   55.57  430.95    94.8  431.77  205.95  431.18  346.52  432.68
   402.1  434.21  451.13   437.3  513.25  444.47  562.28  448.76  657.09  454.41
#Mann= 3 , 0 , 0
 -891.94     .12       0   -9.98    .045       0    9.81     .12       0
#XS Ineff= 2 , 0
          -25.46  437.04
Permanent Ineff=
       F       F
Bank Sta=-9.98,9.81
XS Rating Curve= 0 ,0
Exp/Cntr=0.3,0.1

Type RM Length L Ch R = 1 ,25024.91,434.13,436.44,383.71
XS GIS Cut Line= 3
2447659.24830145331456.3281526862447971.49078719 330236.03794235
2447981.69221036330202.540305942
#Sta/Elev= 30
       0   457.3   98.41  453.64  209.93  447.91  350.98  445.02  413.31  440.88
  442.83  440.19  508.43  441.55  537.96   440.9  551.08  442.34  633.08  436.56
  728.21  427.85  741.33  427.53  748.35  426.07  754.45  425.71  768.21  427.23
  783.97  428.08  843.02  428.06  872.54  430.47  885.66  433.49  905.34  442.07
  925.02  447.77  934.86  448.11  990.63  455.39 1085.75   462.4 1125.12  463.86
 1154.64  463.63 1197.28  460.55 1256.33  460.63 1285.07  457.99 1294.62  457.97
#Mann= 3 , 0 , 0
       0     .12       0  748.35    .045       0  768.21     .12       0
Bank Sta=748.35,768.21
XS Rating Curve= 0 ,0
Exp/Cntr=0.3,0.1

Type RM Length L Ch R = 1 ,24588.47,506.0794,499.9999,460.9907
XS GIS Cut Line= 3
   2448208.47489    331462.79336   2448182.57599    330872.87886
   2448156.56489    330343.82546
#Sta/Elev= 30
 -590.48  461.52 -426.46  457.85 -380.53   455.9 -291.96  447.39 -259.16  443.13
 -177.14  435.29 -154.18  432.18 -108.26  428.81  -78.73  427.38  -68.89  425.66
   -9.91  421.99       0  421.69   10.19  421.84   22.89  422.88   71.93  429.95
   85.01  432.82  111.17  436.58  209.26  446.53  225.61  447.64  245.23  450.29
  271.39  452.08  281.19  454.03  300.81   456.1  362.94  460.31  382.56  462.45
  425.06  464.78  447.95  466.94  487.19  468.81  500.26  469.98  529.69   470.8
#Mann= 3 ,-1 , 0
 -590.48     .12       0   -9.91    .045       0   10.19     .12       0
Bank Sta=-9.91,10.19
XS Rating Curve= 0 ,0
Exp/Cntr=0.3,0.1

Type RM Length L Ch R = 1 ,24088.47,564.6619,604.0481,542.247
XS GIS Cut Line= 4
   2448810.90545    331983.62697   2448748.79238    331139.94591
   2448603.27496    330900.69606   2448292.50196    330389.74302
#Sta/Elev= 30
-1125.99  457.83-1024.35  449.95 -883.35  443.57 -830.89  439.44  -798.1  435.67
 -732.52  436.88 -578.41  435.24  -565.3  436.52  -548.9  435.39 -493.16  436.69
 -421.02  441.78 -332.49  450.39 -227.93  454.71 -166.06   449.7 -123.73  443.27
  -84.66   434.4  -74.89  433.34  -61.87   428.7  -39.07  422.89   -9.77  417.24
       0  416.13   13.07  416.66   22.88  418.12   49.02  417.93   94.77  420.66
  143.79   429.3  218.95  436.88  339.87  444.89     500  459.99  598.04  467.37
#Mann= 3 , 0 , 0
-1125.99     .12       0   -9.77    .045       0   13.07     .12       0
Bank Sta=-9.77,13.07
XS Rating Curve= 0 ,0
Exp/Cntr=0.3,0.1

Type RM Length L Ch R = 1 ,23484.42,372.0689,395.9521,408.801
XS GIS Cut Line= 5
    2449330.2922    331187.04129   2449270.74442    330914.75082
   2448990.08553    330617.10575   2448829.43297    330446.73011
   2448470.91695    330245.20098
#Sta/Elev= 30
 -691.17  450.73 -566.56  439.47 -520.65   438.2 -468.19  439.43 -366.62  433.24
 -340.44  433.19 -301.17  429.42 -278.26  425.21 -222.62  417.73 -186.62  414.73
  -81.89  413.54  -16.43  414.17   -6.62  411.99    3.16  410.67   16.17  411.12
   29.18  411.75   38.94  414.34   71.46   416.1  156.03  425.79  188.55  427.22
  214.57  425.21   234.1  425.68  296.11  435.54   315.7  440.07  361.39  445.26
  403.83   448.3     443  449.05  495.22  453.11  583.35  463.51  642.11  465.52
#Mann= 3 , 0 , 0
 -691.17     .12       0   -6.62    .045       0   16.17     .12       0
Bank Sta=-6.62,16.17
XS Rating Curve= 0 ,0
Exp/Cntr=0.3,0.1

Type RM Length L Ch R = 1 ,23088.47,516.8025,500,476.356
XS GIS Cut Line= 3
   2449449.64958    331239.12452   2449330.22888    330487.52727
   2449246.06009    329965.80751
#Sta/Elev= 30
 -761.03  455.88 -659.34  447.38 -541.25  434.52 -492.04  432.51  -416.6   435.3
 -360.83  434.74 -337.87  433.52 -298.51  429.76 -193.54  415.24 -134.49  412.43
  -29.52  410.95  -13.12  409.05       0  407.24    6.52  408.86   61.98  414.17
    94.6  421.13  117.44  424.56  133.75  429.81  179.42  431.53  192.47  431.18
  198.99  432.67  218.56  433.77  287.07  435.12  332.74  439.07  391.46  441.84
  397.98  443.39  411.03  444.02  450.17  444.66  492.58   446.9  528.47  446.36
#Mann= 3 , 0 , 0
 -761.03     .12       0  -13.12    .045       0    6.52     .12       0
Bank Sta=-13.12,6.52
XS Rating Curve= 0 ,0
Exp/Cntr=0.3,0.1

Type RM Length L Ch R = 1 ,22588.47,474.5533,500,520.5178
XS GIS Cut Line= 4
   2449861.97618    330987.38847    2449926.9872    330411.24035
   2449659.20985    330165.41243   2449108.93799    329672.28415
#Sta/Elev= 30
 -943.31  463.09    -809  455.77  -674.7  445.55 -569.88   443.9 -497.81  439.99
 -412.64  430.33 -347.13  417.75 -275.08  413.59 -229.24  405.75  -22.92  403.93
   -9.82  402.17       0  399.23   13.08  400.71   19.62  403.58   39.23  405.72
  196.17  407.57  228.86  411.51  274.64  420.83  294.25  421.07  320.41  416.78
  340.03  415.75  372.72  415.91  480.61  425.58  493.69  427.39  529.65  437.52
  588.51  449.18  617.93  456.59  647.36  461.16  706.21  466.85   738.9  467.51
#Mann= 3 , 0 , 0
 -943.31     .12       0   -9.82    .045       0   13.08     .12       0
Bank Sta=-9.82,13.08
XS Rating Curve= 0 ,0
Exp/Cntr=0.3,0.1

Type RM Length L Ch R = 1 ,22088.47,522.0925,499.9998,475.454
XS GIS Cut Line= 3
   2450145.83027     331237.3883   2450067.78351     329972.7468
   2450034.60543    329475.15495
#Sta/Elev= 30
-1267.05  439.92   -1159  431.82-1077.15  428.42 -988.76  427.44 -867.62  422.77
 -717.01  419.49 -514.02  430.35 -458.36  431.21 -405.98  426.47 -356.87  418.67
 -337.22  413.71  -327.4  409.52 -304.48  402.69 -225.91  399.08  -72.03  398.01
  -22.92  399.85  -10.09  399.11   -3.27  395.65    3.26  396.04      10   398.5
   22.82  407.01   29.33  409.06   45.63  411.07   97.78  425.57  123.86  431.08
  172.75  440.44  195.57  443.58   257.5  449.02  325.95   451.4   498.7  461.35
#Mann= 3 ,-1 , 0
-1267.05     .12       0  -10.09    .045       0      10     .12       0
Bank Sta=-10.09,10
XS Rating Curve= 0 ,0
Exp/Cntr=0.3,0.1

Type RM Length L Ch R = 1 ,21588.47,491.2853,500,497.9432
XS GIS Cut Line= 3
   2451232.63584    330535.99961   2450521.21272    329896.45562
   2450119.06097    329536.65844
#Sta/Elev= 30
 -956.63  441.53 -835.41  430.52 -743.68  424.19 -632.29  414.11 -540.56  410.68
 -380.03  397.42 -183.46  392.95  -65.52   392.2   -9.83  394.38   -6.55  393.32
       0  390.76    6.54  391.11   13.08  393.66   16.35  394.51    32.7  395.07
   45.78  398.29   71.95  400.54   85.03  404.99  114.46  412.46  130.81  413.42
  156.98  416.81  192.95  424.41  206.03  425.89  238.74   431.5  294.33  442.53
  330.31  447.62  376.09  453.39  438.23  458.65  490.56  461.71  539.61  462.88
#Mann= 3 , 0 , 0
 -956.63     .12       0   -6.55    .045       0   13.08     .12       0
Bank Sta=-6.55,13.08
XS Rating Curve= 0 ,0
Exp/Cntr=0.3,0.1

Type RM Length L Ch R = 1 ,21088.47,423.75,482.85,483.79
XS GIS Cut Line= 5
2451324.64976327330167.9439184372450932.15678185 329681.97573027
2450896.30580369329653.4419946822450861.41020419329626.854449436
2450570.09057686329260.828934774
#Sta/Elev= 30
       0  435.61   35.98  433.31   81.76  428.91  160.26  419.19  215.86  413.43
  248.56  409.02  281.27  403.44  307.43  397.66  327.05  394.93  349.95  393.01
  379.38  391.51  444.79  391.38   477.5  389.68  549.45  389.09  562.53  389.68
  611.59  389.02  644.31  389.86  659.45  391.02  663.95  390.75  673.63  388.24
  680.28  389.26  689.29  392.23  698.69  392.84  737.26  392.78  773.25   394.6
  841.95  399.99  946.63  405.53 1015.33  410.03 1090.57  412.41 1182.17  418.04
#Mann= 3 , 0 , 0
 -669.47     .12       0  659.45    .045       0  680.28     .12       0
Bank Sta=659.45,680.28
XS Rating Curve= 0 ,0
Exp/Cntr=0.3,0.1

Type RM Length L Ch R = 1 ,20605.62,1059.618,1101.115,1069.352
XS GIS Cut Line= 5
2451464.38111112 329887.703993352451247.26081043329520.951446027
2451243.39139561329433.3371199372451237.27821887329345.170301527
2451014.22912428328960.232423097
#Sta/Elev= 30
       0  417.21   49.18  413.55   95.08  408.71  163.92  402.68  193.43  401.17
   213.1  398.85  275.39   393.8  288.51  391.57  324.57  388.78   380.3  387.05
  474.92   387.5  491.17  387.09  504.27  384.84  507.41   384.7  523.31  386.76
  549.91  388.12  612.09  387.88  651.35  391.69  670.98  396.34  680.79  397.98
  703.69  404.36   759.3  418.32  769.12  422.07  792.01     427   805.1  429.11
  841.08  434.02  913.05   438.1  978.48  446.07 1014.46  447.75 1047.17   450.2
#Mann= 3 , 0 , 0
       0     .12       0  504.27    .045       0  523.31     .12       0
Bank Sta=504.27,523.31
XS Rating Curve= 0 ,0
Exp/Cntr=0.3,0.1

Type RM Length L Ch R = 1 ,20054.82,447.9204,466.3531,479.5653
XS GIS Cut Line= 3
   2451838.01882    329852.91043   2451693.06537    329282.75671
   2451553.42162    328771.74035
#Sta/Elev= 30
 -589.96  417.65 -547.47   414.8  -472.3  405.22 -433.08  398.87 -380.79  393.19
 -344.84  390.57 -161.82  384.86  -63.77  384.85  -18.01  385.71  -10.11  383.88
   -4.94  381.96   -1.67  381.48      10  383.82   21.22  385.15   50.65  384.43
   89.89  385.25  112.78  386.89  125.86   388.7  145.48  392.92  174.91  397.52
  201.07  402.48  223.96  407.64  246.85  415.16  276.29  420.46  390.74  429.06
  413.63  430.31  433.25  433.76  469.22  435.33  505.19  438.12  528.08  440.65
#Mann= 3 ,-1 , 0
 -589.96     .12       0  -10.11    .045       0      10     .12       0
Bank Sta=-10.11,10
XS Rating Curve= 0 ,0
Exp/Cntr=0.3,0.1

Type RM Length L Ch R = 1 ,19588.47,987.8606,991.1049,991.9768
XS GIS Cut Line= 4
   2451946.88638    329852.22637   2452113.62686    329286.02245
   2452231.76245    328891.50651   2452090.98353    328093.54584
#Sta/Elev= 30
 -590.25  421.12 -521.38  416.38 -390.22  396.83 -324.63  390.78 -147.56  383.55
  -19.67  383.87  -13.12  382.82   -6.56  380.96       0  380.82    9.81  383.63
   124.2  383.36  150.35  384.35  313.77  397.15  349.72  401.92   372.6  403.66
  451.19  405.33  464.31  403.51  483.99  406.17  506.96  406.09  579.13  408.88
  625.06  412.53   667.7   418.6  697.23  420.11  723.47  419.46   802.2  413.99
  926.86  418.62  956.39  418.68 1067.92  410.36 1159.78  414.04 1222.11  415.24
#Mann= 3 ,-1 , 0
 -590.25     .12       0  -13.12    .045       0   10.14     .12       0
Bank Sta=-13.12,9.81
XS Rating Curve= 0 ,0
Exp/Cntr=0.3,0.1

Type RM Length L Ch R = 1 ,19002.89,406.6,405.53,404.75
XS GIS Cut Line= 3
2452481.72258036329958.7012266812452657.57065386329471.594917431
2453018.37439419 328524.77397643
#Sta/Elev= 30
       0  418.59   45.89  414.93  111.44  411.92  235.99  404.63  285.16  399.54
  347.44  391.82  419.54  384.38   455.6  381.95  491.65  382.51  494.93  382.13
  500.66  379.87  504.77  379.23   514.6  379.57   520.6  381.19  530.99  382.58
  596.57  382.02  986.79  384.02 1085.16  388.11 1121.23   391.2 1131.07  392.86
 1180.25  398.13 1216.32  400.41 1262.23  402.35 1317.97  406.13 1331.09   404.2
 1357.32  405.25 1396.67  407.76 1426.18  408.62 1472.09  413.43 1531.11   415.2
#Mann= 3 , 0 , 0
       0     .12       0  500.66    .045       0   520.6     .12       0
Bank Sta=500.66,520.6
XS Rating Curve= 0 ,0
Exp/Cntr=0.3,0.1

Type RM Length L Ch R = 1 ,18597.36,983.5831,1011.305,1006.18
XS GIS Cut Line= 3
   2452488.99422     331331.4908   2453032.29661    329624.81115
   2453428.66458    328492.08113
#Sta/Elev= 30
-1792.66  411.07-1759.86   410.8-1730.34  408.32-1582.72  405.54-1444.95  408.42
-1307.17  406.84-1228.44  402.77-1139.87  394.43-1070.99  393.54 -946.33  398.76
 -897.13  398.65 -884.01  399.53 -867.61  402.85 -697.03  405.57 -677.35  403.77
 -611.74  401.98 -398.52  385.52   -50.8  381.67  -10.06  379.17    1.55  378.52
   10.05   379.1   24.64  381.03   139.4   380.5  637.79  387.77  952.57  399.26
 1037.82  405.26 1073.89  408.95 1093.56     413 1132.91  416.46 1198.48  417.68
#Mann= 3 ,-1 , 0
-1792.66     .12       0  -10.06    .045       0   10.05     .12       0
Bank Sta=-10.06,10.05
XS Rating Curve= 0 ,0
Exp/Cntr=0.3,0.1

Type RM Length L Ch R = 1 ,18061.84,470.52,475.78,476.28
XS GIS Cut Line= 5
2453605.89257611 331002.671251612453383.54361136330101.025089026
2453480.77307568329801.3908457762453635.92368403329323.259584188
 2453866.3093781328837.740870193
#Sta/Elev= 30
       0  427.42  183.12  425.74     206  426.93  225.62  425.33  317.18  423.52
  519.92   423.3  732.46  416.94  846.91  415.09  863.26  415.52  928.66  411.74
  990.36   411.9 1022.84  411.01 1091.04  405.81 1139.75  398.85 1152.74  395.44
 1178.72  384.56 1188.46  381.41 1227.42  377.32 1248.58   378.1 1253.47  379.79
 1495.01  379.89 1645.16  386.04 1779.12  384.92 1877.42  387.81  1923.3  391.33
 1946.24  394.74 1962.62  398.32 2126.46  416.12 2244.43  425.01 2283.75  425.58
#Mann= 3 , 0 , 0
       0     .12       0 1227.42    .045       0 1248.58     .12       0
Bank Sta=1227.42,1248.58
XS Rating Curve= 0 ,0
Exp/Cntr=0.3,0.1

Type RM Length L Ch R = 1 ,17586.06,532.2178,543.4628,553.2307
XS GIS Cut Line= 3
   2453695.30217    330488.78252   2453878.99308    330018.75688
   2454283.84398     329000.9351
#Sta/Elev= 30
 -605.45  426.11 -553.02  420.76 -477.65  414.75 -412.11  407.37 -362.95     404
  -271.2  401.54 -225.32  402.11 -205.66  404.88 -182.72  405.62 -136.85  403.85
 -123.74  402.06  -64.73  382.66  -45.05  379.66  -22.09  378.36  -15.53  376.85
   -8.97  375.37     .87  376.33   10.71  378.92   86.14  378.17  299.31  379.72
  335.38  380.95  361.62  383.37  453.45  386.37  522.32  391.11  574.79  395.93
  594.47  398.84  610.87   399.7  666.62  407.81  892.92  419.47  994.58  425.72
#Mann= 3 , 0 , 0
 -605.45     .12       0  -15.53    .045       0     .87     .12       0
Bank Sta=-15.53,0.87
XS Rating Curve= 0 ,0
Exp/Cntr=0.3,0.1

Type RM Length L Ch R = 1 ,17042.6 ,518.2399,526.295,526.4755
XS GIS Cut Line= 3
   2453782.76952    330886.35554    2454387.5754    330156.42754
   2454759.88535    329754.97165
#Sta/Elev= 30
 -947.94  420.96 -826.58  412.72 -760.97  409.25 -695.37  407.35 -574.01  402.35
 -469.05  402.01 -364.09  405.23 -341.13  407.66 -328.01  407.79 -301.77  406.46
 -272.24  403.78 -209.92  389.66 -160.72  380.63  -147.6  379.73   -32.8  377.64
  -19.68  375.21   -6.56  374.47     .77  376.15    6.56   377.2  121.31  376.92
  177.04  377.85  206.55  381.92  232.78  387.04  259.01  393.66  291.79   399.3
  334.42  402.29  396.71  409.28  468.84   415.5  514.74  418.05  547.52   418.2
#Mann= 3 ,-1 , 0
 -947.94     .12       0  -19.68    .045       0     .77     .12       0
Bank Sta=-19.68,0.77
XS Rating Curve= 0 ,0
Exp/Cntr=0.3,0.1

Type RM Length L Ch R = 1 ,16516.3 ,467.5559,467.5835,465.4793
XS GIS Cut Line= 5
   2454590.14815    330875.85195   2454641.22154    330562.10455
   2454797.41677    330420.47261   2455009.96162    330227.74498
   2455574.52315    330063.35194
#Sta/Elev= 30
  -512.8  424.04 -326.01  418.61 -303.07  416.37 -237.53  413.55 -194.93  407.67
 -139.78  396.15 -110.59   389.4  -97.61  383.99  -74.91  377.59  -55.44  375.53
     -23  375.87  -16.52     374   -6.79  371.93    6.19  374.06   35.48  376.45
   55.05  374.01  103.95  375.15  113.73  377.31   165.9  383.31  240.89  397.04
  377.97  413.56  430.24  415.53  456.37  411.18   482.5  414.06  538.04  413.56
  567.44  414.88  662.17  422.64  724.24  423.66  786.31  428.63  890.84  432.15
#Mann= 3 , 0 , 0
  -512.8     .12       0  -16.52    .045       0    6.19     .12       0
Bank Sta=-16.52,6.19
XS Rating Curve= 0 ,0
Exp/Cntr=0.3,0.1

Type RM Length L Ch R = 1 ,16048.72,561.5841,579.9158,589.2054
XS GIS Cut Line= 3
   2454743.11241    331097.70912   2455107.05952    330751.14321
   2455472.52336    330403.13308
#Sta/Elev= 30
 -450.71  422.54 -365.86   418.1  -300.6  412.28 -254.91   410.8 -235.33  411.28
 -179.85   403.9 -157.01  398.86 -147.22  396.38 -124.37  388.69 -114.58  384.07
 -101.53  379.12  -78.69  373.67  -62.37  373.22  -19.95  374.41   -9.94  372.74
   -3.63  371.96    6.16  372.03   10.01  373.49   12.69  374.17   45.32  374.24
   68.23  375.21  133.77  381.15   215.7  391.62  271.41  399.59  340.22  404.96
  366.44  407.63  405.76  413.32  418.87  416.53  500.79  419.78   556.5   422.7
#Mann= 3 ,-1 , 0
 -450.71     .12       0   -9.94    .045       0   10.01     .12       0
Bank Sta=-9.94,10.01
XS Rating Curve= 0 ,0
Exp/Cntr=0.3,0.1

Type RM Length L Ch R = 1 ,15468.8 ,385.0684,380.3336,370.2084
XS GIS Cut Line= 3
   2454730.33915    331447.49549   2455377.29717    331225.24331
   2456126.17231     330968.3288
#Sta/Elev= 30
    -690  426.05 -549.26  420.41  -447.8  413.28 -356.15  410.63 -320.15  410.64
 -303.78  407.11 -280.87  404.53 -261.23  401.03  -228.5  397.63 -218.68  393.59
 -182.68  384.66 -140.13  376.11  -94.31  373.17  -51.76  371.95  -19.03   372.7
  -12.48  371.32     .61  370.03    7.15  371.42   13.69  374.52   20.24  376.23
   72.58  378.38   92.21   380.3  141.29   391.2  190.36  394.06  278.69  405.15
  353.94  411.58  422.64  416.06  488.07  417.81  573.13  418.25  785.78  427.45
#Mann= 3 , 0 , 0
    -690     .12       0  -12.48    .045       0    7.15     .12       0
Bank Sta=-12.48,7.15
XS Rating Curve= 0 ,0
Exp/Cntr=0.3,0.1

Type RM Length L Ch R = 1 ,15088.47,478.392,469.1619,451.1669
XS GIS Cut Line= 3
   2455047.78339    331847.32639   2455465.27764    331574.83185
   2455925.21996    331274.63101
#Sta/Elev= 30
 -498.55  423.84 -462.47  421.96 -373.91  414.23 -314.88   410.6 -291.92  404.54
  -262.4  402.39 -239.44  399.15  -229.6  396.82 -173.84  393.64    -164  389.45
 -154.16  386.91  -131.2  383.17 -108.24  378.07  -55.76  373.11  -29.52  372.14
  -22.96  370.38  -13.12  369.53   -3.28  369.08    6.54  369.94   22.89  371.48
   62.12  371.34   81.73  373.06  104.62  375.96  150.39  385.43  179.81  390.23
  264.81  401.69   330.2  408.75  382.51  412.83  441.36  415.76  549.24   417.5
#Mann= 3 , 0 , 0
 -498.55     .12       0  -13.12    .045       0    6.54     .12       0
Bank Sta=-13.12,6.54
XS Rating Curve= 0 ,0
Exp/Cntr=0.3,0.1

Type RM Length L Ch R = 1 ,14619.31,975.3208,1021.72,1039.241
XS GIS Cut Line= 3
   2455535.83294    332291.14768   2455785.29767    331832.88383
   2456043.39361    331358.76503
#Sta/Elev= 30
 -530.79  416.25 -426.44  408.49 -393.83  404.48 -384.04  404.13 -309.04  396.15
 -207.95  388.59 -175.34  385.09 -123.16  377.78  -93.81  375.52  -80.77  372.56
  -25.33  369.97  -12.29  366.79   -5.75  366.27    7.33  367.09   13.88  367.92
   20.42  370.19   23.69  370.53   98.94  371.02  118.57  372.47  174.18  378.94
  203.63  380.95  288.69  391.09  311.59  392.93  318.14  391.89  337.77  393.58
  373.75  395.24   403.2  400.86   426.1  402.35  455.54  407.05  530.79  412.99
#Mann= 3 , 0 , 0
 -530.79     .12       0  -12.29    .045       0    7.33     .12       0
Bank Sta=-12.29,7.33
XS Rating Curve= 0 ,0
Exp/Cntr=0.3,0.1

Type RM Length L Ch R = 1 ,14017.4 ,415.81,419.81,419.35
XS GIS Cut Line= 3
2455678.46192178332180.6429770142456148.34746495332132.138480857
 2456647.2116247332080.641864687
#Sta/Elev= 30
       0   405.1   22.96  404.57   65.61  402.15  154.18  393.55  177.14  390.11
  255.87   382.1  288.68  380.06   301.8  378.33  314.92  373.62  321.48  372.31
  344.45  369.85  410.05  367.88  442.86  368.22  462.25  365.52  465.82  365.22
  472.38  365.67  483.09  367.76  495.33  369.98  505.16  372.71  547.77  387.19
  577.27  399.32  593.66  403.45  606.78  404.71  636.28  409.54  711.67  419.17
  734.61  421.86  754.28  423.19  796.89  428.33  885.39  435.32   973.9  439.16
#Mann= 3 , 0 , 0
       0     .12       0  462.25    .045       0  483.09     .12       0
Bank Sta=462.25,483.09
XS Rating Curve= 0 ,0
Exp/Cntr=0.3,0.1

Type RM Length L Ch R = 1 ,13597.59,521.0212,509.1174,491.5662
XS GIS Cut Line= 4
   2455560.63375    332565.64221   2456073.70194    332532.07403
   2456429.72518    332508.78044   2456635.57648    332221.58122
#Sta/Elev= 30
 -627.41  426.45 -591.39  424.25 -480.04  411.64 -434.19  409.02 -398.16   404.7
 -355.59  401.43 -313.02  394.01 -254.07  387.73 -237.69  382.95 -224.59  381.02
 -211.49  381.74 -188.57  373.47 -168.92  368.68 -103.43  366.08  -64.15  366.13
  -15.05  368.01    -8.5  364.79   -5.23  364.66   10.26  367.17   63.51  368.77
  112.61  374.92  128.98  375.77  184.62  384.57  214.08  385.25  302.43  393.23
   387.5  398.16  456.21  404.14  472.56  406.45  518.37  409.34  596.89  417.22
#Mann= 3 , 0 , 0
 -627.41     .12       0  -15.05    .045       0   10.26     .12       0
Bank Sta=-15.05,10.26
XS Rating Curve= 0 ,0
Exp/Cntr=0.3,0.1

Type RM Length L Ch R = 1 ,13095.93,981.4587,1007.46,1016.131
XS GIS Cut Line= 4
2455833.18667795333228.7501327692456273.36886844332967.681757271
2456606.18349153332770.2920601822456849.47204694332766.755649939
#Sta/Elev= 30
       0  416.44  108.26  411.88  164.03  408.01  180.43  404.68  249.33  396.67
  298.54  388.81  337.91  384.72  380.55  378.98  429.76  375.94  459.29   372.5
  465.85  372.55  482.25  368.61  492.09  364.26  497.05  363.45  505.22   362.9
  517.51  364.51  551.13  366.28  597.04   365.6   682.3  369.23  705.25  372.54
  741.32  380.15  767.56   383.3  793.79  385.14  806.91  388.75  934.41  399.32
 1002.54  402.89  1051.2  404.15  1080.4  406.69 1129.06  407.71 1142.04  406.82
#Mann= 3 , 0 , 0
       0     .12       0  497.05    .045       0  517.51     .12       0
Bank Sta=497.05,517.51
XS Rating Curve= 0 ,0
Exp/Cntr=0.3,0.1

Type RM Length L Ch R = 1 ,12588.47,499.4636,499.9999,490.1347
XS GIS Cut Line= 3
   2455900.71115    333526.04416   2456383.34371    333400.92827
   2457047.03464     333229.3935
#Sta/Elev= 30
 -498.59  418.47 -383.78  418.71 -344.42  418.03 -318.18  416.16 -275.53  410.59
 -200.09  403.09 -150.89  392.95  -85.28  380.64  -39.36  370.88  -26.24  363.36
  -22.96  362.05   -16.4  361.59   -3.28   360.1    3.28  362.33    9.84  364.93
   131.2  366.15  196.79  369.05  219.75  371.85  232.87  375.23  262.39  377.32
  298.47   381.8  360.79  384.98  393.59  388.44  465.75  390.28  528.06  390.36
  544.46   389.5  577.26  391.41  600.22  391.23   636.3  392.66   685.5  391.58
#Mann= 3 ,-1 , 0
 -498.59     .12       0   -16.4    .045       0    3.28     .12       0
Bank Sta=-16.4,3.28
XS Rating Curve= 0 ,0
Exp/Cntr=0.3,0.1

Type RM Length L Ch R = 1 ,12088.47,496.2543,500,502.5456
XS GIS Cut Line= 3
   2456199.42676    334021.26823   2456651.27658    333784.83268
   2457094.47254    333552.92534
#Sta/Elev= 30
 -417.86  407.66 -352.48  408.07 -326.33  407.42  -287.1   405.1 -257.68  402.12
 -241.34  398.81 -221.72  396.44 -211.91   394.1 -202.11  393.36 -169.42  386.78
 -120.38  378.93  -84.42  372.08  -28.85     366  -22.31  362.43  -15.77  361.71
   -2.69  359.54    3.84  360.29    7.11  361.86   10.38  363.74   16.92   364.4
    82.3  364.59  121.53  366.15  147.69  370.33   167.3  375.95  173.84  377.06
  255.57  385.06  314.42  389.88  396.15  392.72  520.39  401.84  592.31  405.11
#Mann= 3 , 0 , 0
 -417.86     .12       0  -15.77    .045       0    7.11     .12       0
Bank Sta=-15.77,7.11
XS Rating Curve= 0 ,0
Exp/Cntr=0.3,0.1

Type RM Length L Ch R = 1 ,11588.47,461.0393,469.1768,474.1958
XS GIS Cut Line= 3
   2456450.03813    334401.20481   2456912.82724    334216.66712
   2457395.90501    334024.03922
#Sta/Elev= 30
 -301.88  407.45  -239.6  407.92 -154.37  402.43 -128.15  399.01  -88.82  389.86
  -78.99  385.84  -39.65  372.78   -33.1  371.33  -13.43  364.23   -9.98  363.66
    -3.6  358.78    2.96  358.32    6.24  358.98   12.79  362.65   52.13  361.46
   173.4  365.18  183.24   366.1  206.16  369.83  317.37  376.24  395.87  385.27
  418.77  386.49  428.58  388.17  438.39  388.27  474.37  390.86  497.27  390.72
  539.79  394.01  615.02  397.77  660.81  398.75  677.17  400.13  716.42  399.95
#Mann= 3 , 0 , 0
 -301.88     .12       0   -9.98    .045       0   12.79     .12       0
Bank Sta=-9.98,12.79
XS Rating Curve= 0 ,0
Exp/Cntr=0.3,0.1

Type RM Length L Ch R = 1 ,11119.29,520.8438,530.8229,522.9866
XS GIS Cut Line= 3
   2455920.73243    334888.42135   2456915.93911    334697.75572
   2457517.95496    334610.64369
#Sta/Elev= 30
-1013.31  417.28 -947.72  403.88 -901.81  398.28 -849.34     394 -734.57  387.48
 -685.38  382.59 -646.02  376.55 -547.64  373.75 -511.57   376.2 -485.34   376.3
 -357.44  385.12 -278.74  385.53 -203.32  387.73 -170.52  386.59 -127.89  383.09
   -78.7  373.59  -49.19  365.89  -26.23  363.96   -16.4  359.95  -13.12  357.67
   -6.56  356.76   -3.28  356.93    3.27  359.98  163.52  362.82  179.87  365.08
   209.3  372.21  281.25  381.63  330.31  386.47  490.55  396.65  608.29  396.83
#Mann= 3 , 0 , 0
-1013.31     .12       0   -16.4    .045       0    3.27     .12       0
Bank Sta=-16.4,3.27
XS Rating Curve= 0 ,0
Exp/Cntr=0.3,0.1

Type RM Length L Ch R = 1 ,10588.47,483.8662,500.0002,512.3649
XS GIS Cut Line= 3
   2456535.97399    335246.17162   2457040.95067    335142.21251
   2457748.85772    334997.36241
#Sta/Elev= 30
 -515.57  390.79 -414.41  391.59 -345.89  389.98 -303.47   387.5 -254.52  380.77
 -241.47  377.28 -156.63  362.08 -117.47  360.38 -107.68  358.85  -22.84  359.32
  -16.32  357.57  -13.05  355.57   -9.79  354.92   -3.26  355.64    3.27  357.98
    9.81  359.15   39.23   360.6   91.55  361.45   117.7  363.31  173.29  371.61
  205.98  374.87   225.6  377.95  274.64   381.7  313.88  382.24  353.11  380.56
  382.54  382.15  405.43  381.78  461.01  384.23  575.44  393.04  722.57  399.96
#Mann= 3 , 0 , 0
 -515.57     .12       0  -16.32    .045       0    3.27     .12       0
Bank Sta=-16.32,3.27
XS Rating Curve= 0 ,0
Exp/Cntr=0.3,0.1

Type RM Length L Ch R = 1 ,10088.47,513.2407,500,484.5606
XS GIS Cut Line= 3
   2456302.85076    335451.52915   2457008.73387    335627.37657
   2457528.11111    335761.42486
#Sta/Elev= 30
 -727.46  389.33 -648.81  381.55 -609.49  379.29 -566.89  379.41 -553.78  378.17
  -494.8  378.87 -393.22   372.3 -281.81   369.3 -199.89  361.44 -154.01  359.31
  -140.9  356.13  -127.8  357.63 -108.14  356.05  -52.43  355.88  -22.94  356.78
  -16.38  356.46  -13.11  354.72   -6.55  352.77       0  353.73    3.27  355.46
    9.81  356.66   49.06   357.2   68.69  359.39  117.75  367.83  150.45  371.39
  343.42  385.82  438.28  397.09   457.9  396.77  480.79  401.63   536.4  402.48
#Mann= 3 , 0 , 0
 -727.46     .12       0  -13.11    .045       0    3.27     .12       0
Bank Sta=-13.11,3.27
XS Rating Curve= 0 ,0
Exp/Cntr=0.3,0.1

Type RM Length L Ch R = 1 ,9589.33 ,1401.094,1473.954,1502.972
XS GIS Cut Line= 4
2456509.30573252336239.2480487672456938.42823386336141.882429853
 2457111.1713267335996.0490601062457556.75704969335796.581283182
#Sta/Elev= 30
       0   424.8   88.01  421.92  117.34  423.09  143.42  422.58  237.94  413.73
  254.24  410.01  296.61  403.79  309.65  400.11  319.43  395.64   378.1  378.23
  391.14  372.84  413.95  366.67  443.31   362.3  476.07  355.56  492.45  355.22
  508.83  353.44  521.94  353.82  527.82  352.46  531.77  351.93  548.06  354.25
   597.3   354.1  652.99  355.86  715.25  362.76  744.74   367.8  820.09  378.15
  843.03  379.18  872.52  383.35 1059.28  397.63 1134.63  400.67 1154.29  399.98
#Mann= 3 , 0 , 0
       0     .12       0  527.82    .045       0  548.06     .12       0
Bank Sta=527.82,548.06
XS Rating Curve= 0 ,0
Exp/Cntr=0.3,0.1

Type RM Length L Ch R = 1 ,9101.002,996.1848,1015.216,1021.92
XS GIS Cut Line= 5
2456510.55737044 336291.157065692456945.37277378336493.445046932
2457068.32823652336494.1031821072457204.05335878336493.445046932
2457543.18096136336666.879083276
#Sta/Elev= 30
       0  422.67   48.94  419.95  110.92  412.84     199  408.72  247.94  403.31
  267.51  400.65  290.35  394.94  319.71  392.61   329.5  389.82  401.27  376.17
  414.32  375.31   518.4  354.48  537.81  352.67   573.4  352.33  590.81  349.85
  592.82   349.8  599.29  351.82  609.31  352.52  699.47  353.14  741.51  360.71
  783.83  362.59  806.62  374.27  842.43  383.66   852.2  387.84  865.22  390.45
  878.24  394.98  920.56  404.14  982.42  414.44  1086.6  427.59 1119.15  429.62
#Mann= 3 , 0 , 0
       0     .12       0  590.81    .045       0  609.31     .12       0
Bank Sta=590.81,609.31
XS Rating Curve= 0 ,0
Exp/Cntr=0.3,0.1

Type RM Length L Ch R = 1 ,8600.162,536.93,511.69,476.84
XS GIS Cut Line= 5
2456297.48266536336411.5282160192456691.57669345336715.683775693
 2456736.7941227336781.7400740242456789.23266611336874.104062527
2457123.63061936337101.726966858
#Sta/Elev= 30
       0  419.28  163.76     411  281.66  400.63  304.58  399.16  334.06  398.82
  353.71  394.64  406.11  387.09  415.94  383.65  432.31  381.31  513.83  364.61
  529.84  359.35  542.64  356.73  566.02  349.97  574.66  348.58  587.94  350.35
   600.4  351.02  613.27  349.82  639.02   351.3  674.42  358.41  693.86  360.36
  723.23  365.42  759.11  373.33  781.95  376.81  804.78   382.9  866.76  391.83
  879.81  392.96   889.6  395.32  932.01  401.58 1023.35  410.69 1088.59  415.29
#Mann= 3 , 0 , 0
       0     .12       0  566.02    .045       0  587.94     .12       0
Bank Sta=566.02,587.94
XS Rating Curve= 0 ,0
Exp/Cntr=0.3,0.1

Type RM Length L Ch R = 1 ,8088.469,512.9053,499.9999,482.1624
XS GIS Cut Line= 3
    2455986.0161    337170.33083   2456484.44653    337188.93414
   2457144.25689     337213.5604
#Sta/Elev= 30
 -498.78  414.81  -423.8  411.09 -414.02  409.66 -381.42  407.47 -280.36  396.45
  -244.5  393.21 -172.78  383.85 -153.22  379.94 -127.14  372.24   -97.8  359.35
  -88.02  354.45   -81.5  352.18  -58.68  349.78   -16.3  348.09  -13.04  346.77
   -9.78  344.87       0  344.37    6.54  346.56   29.42  351.83   45.76  352.63
    62.1  354.37   114.4  363.66  176.51  372.32  254.96  382.66  395.51   399.2
  477.22   406.5  532.79  408.76  578.55  412.85  611.24   412.9  660.27   415.2
#Mann= 3 , 0 , 0
 -498.78     .12       0  -13.04    .045       0    6.54     .12       0
Bank Sta=-13.04,6.54
XS Rating Curve= 0 ,0
Exp/Cntr=0.3,0.1

Type RM Length L Ch R = 1 ,7588.469,977.0941,988.7577,993.7749
XS GIS Cut Line= 3
   2455825.31596      338044.897   2456635.83993    337630.28923
   2457253.70123    337309.21999
#Sta/Elev= 30
 -910.41  410.23 -858.01  408.92 -713.92  396.07 -681.17  396.23  -520.7   385.4
 -468.31  378.56 -425.73  375.22 -415.91  373.09 -383.16  371.73 -347.14  367.97
 -330.76   368.3 -245.61  362.39 -199.77  362.59 -193.22  361.04 -170.29  360.73
 -144.09  356.94 -121.17  350.54 -108.07  348.73  -29.47  345.89  -16.37  343.77
   -6.55   341.8    6.54  343.82    42.5  350.94   98.07   358.6  124.22  363.64
  251.72  379.37  307.29  382.18   464.2  393.79  594.96  409.64   696.3  418.85
#Mann= 3 , 0 , 0
 -910.41     .12       0  -16.37    .045       0    6.54     .12       0
Bank Sta=-16.37,6.54
XS Rating Curve= 0 ,0
Exp/Cntr=0.3,0.1

Type RM Length L Ch R = 1 ,7063.755,465.86,464.04,459.51
XS GIS Cut Line= 5
2456482.71293794338216.0800531062456923.22813302337845.827184692
2457020.52649486337838.034221277 2457098.2281111337832.285545111
2457520.62851302337434.220068276
#Sta/Elev= 30
       0  410.66   78.47  406.26  232.14  394.18  297.53  386.36   333.5  384.32
  385.81  377.49  474.09  370.88   516.6  364.41  546.02  357.85   559.1  352.21
  588.46  346.12     621  342.63  650.28  341.83  663.05  338.84   669.8  337.07
  683.01   338.8  692.54   341.4     725  355.02  737.99  356.21  744.48   359.5
  777.21  369.62  796.88  373.67  823.11   381.5  875.58  391.67  914.93  396.16
  960.84  404.58 1095.29  417.32 1246.12  424.29 1305.15  424.32 1331.38  426.07
#Mann= 3 , 0 , 0
       0     .12       0  663.05    .045       0  683.01     .12       0
Bank Sta=663.05,683.01
XS Rating Curve= 0 ,0
Exp/Cntr=0.3,0.1

Type RM Length L Ch R = 1 ,6599.711,526.8891,511.2423,494.5436
XS GIS Cut Line= 3
   2456512.30605    338389.68338   2457001.91564     338292.2925
   2457526.26334    338187.99153
#Sta/Elev= 30
 -499.68  409.65 -447.48   408.5 -382.22   403.9 -330.02  396.75 -320.23  396.74
 -316.97  395.79 -258.24  389.18 -228.87  383.91 -215.82  380.47 -160.35  369.57
 -114.68  358.79  -98.36  352.94     -69  346.04  -29.84  342.28  -23.32  342.32
  -20.06  341.69   -9.96  337.47    -.48  335.36   10.07  337.22    35.6  340.07
   71.68   348.9   88.08  354.26  137.28  361.46  163.51  366.37  265.19  376.51
  291.43   378.2  343.91  379.34  363.59  380.51  445.58  390.22  534.14  397.12
#Mann= 3 ,-1 , 0
 -499.68     .12       0   -9.96    .045       0   10.07     .12       0
Bank Sta=-9.96,10.07
XS Rating Curve= 0 ,0
Exp/Cntr=0.3,0.1

Type RM Length L Ch R = 1 ,6088.469,498.3737,500,496.3019
XS GIS Cut Line= 3
   2456820.28116    339116.77215   2457308.30807    338673.49318
   2457747.36461    338281.70263
#Sta/Elev= 30
 -659.29  373.48 -551.05  371.91 -534.65  370.58 -521.53  371.11 -442.81  366.69
 -380.49  364.74 -324.73  358.61 -239.44  353.95 -144.32  345.41  -91.84  337.89
   -16.4  334.01       0   333.3    6.54  334.63   13.08   336.3   26.15  337.22
   39.23  335.98   65.38  343.98   88.27  354.78   98.07  357.67  117.69   362.2
  156.92  367.74  215.76  379.31  232.11  380.19  304.03  390.71  336.72  393.16
  408.64  401.16  457.68  404.56   487.1   405.3  565.56  411.02  588.45  411.62
#Mann= 3 , 0 , 0
 -659.29     .12       0   -16.4    .045       0    6.54     .12       0
Bank Sta=-16.4,6.54
XS Rating Curve= 0 ,0
Exp/Cntr=0.3,0.1

Type RM Length L Ch R = 1 ,5588.469,502.1185,499.9999,495.3267
XS GIS Cut Line= 3
   2457316.79657     339257.1905   2457734.46667    338872.58366
   2458104.13489    338532.17883
#Sta/Elev= 30
 -567.78  393.02 -469.88  389.31 -443.78  389.89 -430.73   387.7  -398.1  386.92
 -352.41  382.79 -290.41  380.92 -231.68  376.77 -202.31  373.05  -150.1  362.67
    -124  356.39  -94.63  344.97     -62  335.94  -22.84   331.1  -10.19   327.7
    3.26  326.85   10.18  326.89   16.32  327.57   29.37  332.25   55.47  335.33
   94.63  352.12  133.79  365.02  176.21  382.37  189.26   385.7  202.31  386.75
  267.58  398.74     310  404.41  427.47  412.58   460.1  416.48  502.52  418.26
#Mann= 3 ,-1 , 0
 -567.78     .12       0  -10.19    .045       0   10.18     .12       0
Bank Sta=-10.19,10.18
XS Rating Curve= 0 ,0
Exp/Cntr=0.3,0.1

Type RM Length L Ch R = 1 ,5088.469,348.2568,345.5603,335.5764
XS GIS Cut Line= 3
   2457547.72721    339700.66206    2457875.7095    339322.92987
   2458248.51715    338893.57345
#Sta/Elev= 30
 -500.25  397.35 -434.86  391.48 -369.47  389.69 -264.84  379.49 -235.41  377.62
 -189.64  372.35 -176.56  369.77 -140.59  367.12  -107.9  361.02  -78.47  347.81
  -62.12  342.13  -39.24  331.68  -10.17  325.39   -3.27  324.35   11.75  325.47
   22.88  328.02   45.75  328.25   65.36  329.77   75.16  331.61  104.57  339.81
   163.4  360.29  202.61  367.44  225.49  374.18  235.29  375.38   264.7  382.97
  294.12  385.78  320.26   390.1  411.76  401.51  486.92  406.96  568.62   410.3
#Mann= 3 ,-1 , 0
 -500.25     .12       0  -10.17    .045       0   11.75     .12       0
Bank Sta=-10.17,11.75
XS Rating Curve= 0 ,0
Exp/Cntr=0.3,0.1

Type RM Length L Ch R = 1 ,4742.909,672.973,654.4398,624.5975
XS GIS Cut Line= 3
   2457690.02253    340078.32469   2458129.42815    339547.27391
    2458465.8471    338976.97912
#Sta/Elev= 30
 -742.85  401.93 -713.45  401.21 -664.45  396.99 -393.32  378.87 -347.58  376.98
 -305.12  378.02 -252.85  375.25 -161.38   358.1 -154.85  355.75 -148.32  350.32
 -135.25  344.08 -112.38   336.3  -99.32  334.91  -86.25  330.48  -76.45  328.67
  -30.64  324.93  -17.53  322.51  -10.97  321.56    5.42  322.45   18.53  324.26
   28.36  329.87   48.03  336.02   61.14  342.75  116.87  359.95  182.42  372.93
  297.15  385.11  359.43  388.98   408.6  389.65  536.43  402.15  608.55  406.55
#Mann= 3 , 0 , 0
 -742.85     .12       0  -17.53    .045       0    5.42     .12       0
Bank Sta=-17.53,5.42
XS Rating Curve= 0 ,0
Exp/Cntr=0.3,0.1
